--- RFMIDDLERV.prj (project) ---

Proj Title=RFMIDDLERV
Current Plan=p01
Default Exp/Contr=0.3,0.1
English Units
Geom File=g01
Flow File=f01
Plan File=p01
Y Axis Title=Elevation
X Axis Title(PF)=Main Channel Distance
X Axis Title(XS)=Station
BEGIN DESCRIPTION:
END DESCRIPTION:
DSS Export Rating Curves= 0
DSS Export Rating Curve Sorted= 0
DSS Export Volume Flow Curves= 0
DXF OffsetX= 0
DXF OffsetY= 0
DXF ScaleX= 1
DXF ScaleY= 10

--- RFMIDDLERV.p01 (plan) ---

Plan Title=Floodplain
Program Version=6.30
Short Identifier=Floodplain
Geom File=g01
Flow File=f01
Subcritical Flow
K Sum by GR= 0
Std Step Tol= 0.01
Critical Tol= 0.01
Num of Std Step Trials= 20
Max Error Tol= 0.3
Flow Tol Ratio= 0.001
Split Flow NTrial= 30
Split Flow Tol= 0.02
Split Flow Ratio= 0.02
Log Output Level= 0
Friction Slope Method= 1
Unsteady Friction Slope Method= 2
Unsteady Bridges Friction Slope Method= 1
Parabolic Critical Depth
Global Vel Dist= 0 , 0 , 0
Global Log Level= 0
CheckData=True
Encroach Param=-1 ,0,0, 0
Computation Interval=1MIN
Output Interval=1HOUR
Instantaneous Interval=1HOUR
Mapping Interval=1HOUR
Computation Time Step Use Courant=        0
Computation Time Step Use Time Series=    0
Computation Time Step Count To Double=0
Computation Time Step Max Doubling=0
Computation Time Step Max Halving=0
Computation Time Step Residence Courant=0
Run HTab= 0
Run UNet= 0
Run Sediment= 0
Run PostProcess= 0
Run WQNet= 0
Run RASMapper= 0
UNET Theta= 1
UNET Theta Warmup= 1
UNET ZTol= 0.02
UNET ZSATol= 0.02
UNET MxIter= 20
UNET Max Iter WO Improvement= 0
UNET MaxInSteps= 0
UNET DtIC= 0
UNET DtMin= 0
UNET MaxCRTS= 20
UNET WFStab= 2
UNET SFStab= 1
UNET WFX= 1
UNET SFX= 1
UNET Gravity=32.17405
UNET 1D Methodology=Finite Difference
UNET DSS MLevel= 4
UNET Pardiso=0
UNET DZMax Abort= 100
UNET Use Existing IB Tables=-1
UNET Froude Reduction=False
UNET Froude Limit= 0.8
UNET Froude Power= 4
UNET D1 Cores= 0
UNET WindReference=Eulerian
UNET WindDragFormulation=Hsu (1988)
UNET D2 Coriolis=0
UNET D2 Cores= 0
UNET D2 Theta= 1
UNET D2 Theta Warmup= 1
UNET D2 Z Tol= 0.01
UNET D2 Volume Tol= 0.01
UNET D2 Max Iterations= 20
UNET D2 Equation= 0
UNET D2 RampUpFraction=0.1
UNET D2 TimeSlices= 1
UNET D2 Turbulence Formulation=None
UNET D2 Eddy Viscosity=0.3
UNET D2 Transverse Eddy Viscosity=0.1
UNET D2 Smagorinsky Mixing=0.05
UNET D2 BCVolumeCheck=0
UNET D2 Cores=0
UNET D2 SolverType=PARDISO (Direct)
UNET D2 Minimum Iterations= 3
UNET D2 Maximum Iterations= 30
UNET D2 Restart Number= 10
UNET D2 Relaxation Coeff=1.3
UNET D2 SOR Precondition Iterations= 10
UNET D2 ILUT Maximum Fill= 8
UNET D2 ILUT Tolerance=1E-08
UNET D2 Convergence Tolerance=0.00001
UNET D1D2 MaxIter= 0
UNET D1D2 ZTol=0.01
UNET D1D2 QTol=0.1
UNET D1D2 MinQTol=1
Write IC File= 0
Write IC File at Fixed DateTime=0
Write IC File at Sim End=0
Echo Input=False
Echo Parameters=False
Echo Output=False
Write Detailed= 0
HDF Write Warmup=0
HDF Write Time Slices=0
HDF Flush=0
HDF Compression= 1
HDF Chunk Size= 1
HDF Spatial Parts= 1
HDF Use Max Rows=0
HDF Fixed Rows= 1
Calibration Method= 0
Calibration Iterations= 20
Calibration Max Change=0.05
Calibration Tolerance=0.2
Calibration Maximum=1.5
Calibration Minimum=0.5
Calibration Optimization Method= 1
WQ AD Non Conservative
WQ ULTIMATE=-1
WQ Max Comp Step=1HOUR
WQ Output Interval=15MIN
WQ Output Selected Increments= 0
WQ Output face flow=0
WQ Output face velocity=0
WQ Output face area=0
WQ Output face dispersion=0
WQ Output cell volume=0
WQ Output cell surface area=0
WQ Output cell continuity=0
WQ Output cumulative cell continuity=0
WQ Output face conc=0
WQ Output face dconc_dx=0
WQ Output face courant=0
WQ Output face peclet=0
WQ Output face adv mass=0
WQ Output face disp mass=0
WQ Output cell mass=0
WQ Output cell source sink temp=0
WQ Output nsm pathways=0
WQ Output nsm derived pathways=0
WQ Create Restart=0
WQ Fixed Restart=0
WQ System Summary=0
WQ Write To DSS=0
Sorting and Armoring Iterations= 10
XS Update Threshold= 0.02
Bed Roughness Predictor= 0
Hydraulics Update Threshold= 0.02
Energy Slope Method= 1
Volume Change Method= 1
Sediment Retention Method= 0
Sediment TS Multiplier= 1
Warm Up Method= 0
XS Weighting Method= 0
Number of US Weighted Cross Sections= 1
Number of DS Weighted Cross Sections= 1
Upstream XS Weight=0
Main XS Weight=1
Downstream XS Weight=0
Number of DS XS's Weighted with US Boundary= 1
Upstream Boundary Weight= 1
Weight of XSs Associated with US Boundary= 0
Number of US XS's Weighted with DS Boundary= 1
Downstream Boundary Weight= 0.5
Weight of XSs Associated with DS Boundary= 0.5
Percentile Method= 0
Sediment Output Level= 3
Mass or Volume Output= 0
Output Increment Type= 1
Profile and TS Output Increment= 1
Transport Output Increment 1
XS Output Flag= 0
XS Output Increment= 10
Read HDF5 Sediment Hotstart= 0
Sediment Hotstart Type= 0
Write Gradation File= 0
Read Gradation Hotstart= 0
Write HDF5 File= 1
Write Binary Output= 1
Write DSS Sediment File= 0
DSS Sediment Output Type= 1
SV Curve= 0
Specific Gage Flag= 0
Subcell Erosion Methods= 0
Subcell Deposition Methods= 0
Advection Scheme= 1
Matrix Solver= 0
Implicit Weighting Factor= 1
Maximum Outer Loop Convergence Iterations= 5
Convergence Maximum Absolute= 0.001
Convergence RMSE= 0.0001
Grain Fractions Max Abs Error= 0.001
Max Subgrid Regions= 1
Max Subgrid Length Scale= 3.402823E+38
Initial Layer Thickness= 3.402823E+38
Min Layer Thickness= 3.402823E+38
Max Layer Thickness= 3.402823E+38
Number of Layers= 5

--- RFMIDDLERV.f01 (steady flow) ---

Flow Title=Flows
Program Version=6.30
Number of Profiles= 1
Profile Names=100Yr
River Rch & RM=River 1,Reach 1         ,77998
     429
River Rch & RM=River 1,Reach 1         ,73982
     680
River Rch & RM=River 1,Reach 1         ,70461
    1100
River Rch & RM=River 1,Reach 1         ,63781
    1280
River Rch & RM=River 1,Reach 1         ,60998
    1430
River Rch & RM=River 1,Reach 1         ,51486
    1590
River Rch & RM=River 1,Reach 1         ,46680
    1770
River Rch & RM=River 1,Reach 1         ,39504
    1970
River Rch & RM=River 1,Reach 1         ,37619
    2920
River Rch & RM=River 1,Reach 1         ,35386
    3580
River Rch & RM=River 1,Reach 1         ,20481
    3980
River Rch & RM=River 1,Reach 1         ,8186
    4550
Boundary for River Rch & Prof#=River 1,Reach 1         , 1
Up Type= 0
Dn Type= 3
Dn Slope=0.0025
DSS Import GetInterval= 0
DSS Import GetPeak= 0
DSS Import FillOption= 0

--- RFMIDDLERV.g01 (geometry) ---

Geom Title=Geometry
Program Version=6.30

River Reach=River 1         ,Reach 1
Reach XY= 30
2219177.73969478643113.7863898192216099.43057276644640.819703758
2216234.69998726647597.3790793422214347.73558535648408.939792171
2214376.66662984649405.9633886672213564.70532726649312.273287341
2213802.36430076652464.3969043342212226.40255767654592.254525259
2212914.94153492656214.4028557542211790.54647401659464.166041255
 2212245.7758785660998.2905976772209844.97523393664781.090774834
 2211706.6430985667256.808920503 2212299.6891565670814.140716583
2214995.32418518  671394.28096052215935.14382784673267.538368836
2214890.55963093675051.283489004 2215378.2975006676475.235037416
2214423.39717942677463.9597660012215271.90171601 679199.11476025
 2213970.6858145680307.7421361662217156.83462593681332.351963595
2216953.51515068 682454.658117922218862.08515242684188.267511591
2218212.06381467686628.1865162552216720.40603684687138.101835012
2215690.04425243688662.9832996732216836.78900617689861.294551343
2216086.03788301    691059.176672222076.56395967691959.104988262

Type RM Length L Ch R = 1 ,77998   ,49.3,41.5,39.5
XS GIS Cut Line= 5
2219260.03424901643012.043316241  2219231.482832643085.423126293
2219201.86407231643098.2312385932219154.10048686643122.513284829
2219132.52245848643216.268517389
#Sta/Elev= 30
       0 2662.77    10.6 2654.45    18.4 2649.77      27 2645.81    39.8 2636.81
    44.1  2635.5    48.4 2634.56    56.4 2634.31    69.9 2636.01    87.2 2635.68
   121.9 2634.83   126.4 2634.44   130.9 2633.47   135.3 2632.31     144 2632.62
   148.8 2633.47   157.8 2636.53   162.3 2636.75   179.6 2636.57   187.8 2635.93
   200.2 2635.75   208.4 2634.03   212.5 2633.57   220.7 2633.54   224.8 2634.71
   228.9 2637.29     233 2639.12   237.1 2640.17   249.4 2642.04   260.8 2642.14
#Mann= 3 ,-1,0
       0      .1       0   130.9    .045       0   148.8      .1       0
Bank Sta=130.9,148.8
XS Rating Curve= 0 ,0
Exp/Cntr(USF)=0,0
Exp/Cntr=0.3,0.1

Type RM Length L Ch R = 1 ,77956   ,190.3,174.7,157.5
XS GIS Cut Line= 6
2219184.03773896642853.8072615142219175.97211892643057.815235375
2219167.80694733643066.460711177 2219157.7205589643074.145578556
2219134.66595676643090.9562259492219104.73287757643229.960042498
#Sta/Elev= 30
       0 2707.36      37 2695.65    51.4 2689.92    59.4 2687.73    68.6 2683.28
    83.4 2681.11    91.4 2677.74    99.4 2676.31   131.5 2668.46   139.5  2665.3
   147.5 2661.14   163.5 2659.06   167.5  2657.7   182.9  2650.1   187.5 2646.96
   203.5 2634.13   205.92633.286   209.2 2632.39   220.6 2633.34   230.7 2632.26
   243.5 2633.51   254.3  2635.2   275.9 2634.74   304.6 2636.38   311.7 2635.53
   320.9 2635.57   329.1 2633.45   349.6  2633.8   374.1 2641.43   399.5 2644.42
#Mann= 3 ,-1,0
       0      .1       0   205.9    .045       0   243.5      .1       0
Bank Sta=205.9,243.5
XS Rating Curve= 0 ,0
Exp/Cntr(USF)=0,0
Exp/Cntr=0.3,0.1

Type RM Length L Ch R = 1 ,77781   ,164.7,182.6,188.6
XS GIS Cut Line= 4
2218983.93199746642843.6610469892218995.72988584642971.325910486
2219018.76151076643287.1881951182218975.61712295643409.704932345
#Sta/Elev= 30
       0 2683.55     5.5 2680.16    10.3 2678.73    29.6  2677.9    37.7 2678.21
    45.7 2676.18    53.7  2672.9    85.5 2665.24   138.1 2654.03   158.1  2647.3
   182.2 2644.62   198.9 2638.15   214.3 2633.44   246.5 2632.26   282.5 2631.73
   287.4 2632.58   291.1 2633.85   310.5 2634.94   330.6  2631.8   362.7 2632.38
   393.6 2641.63   406.8 2644.22   430.9 2647.04   444.9 2647.73     461 2647.55
   492.4 2651.95     525 2653.93   544.6 2656.68   561.8 2659.83   574.8 2662.97
#Mann= 3 ,-1,0
       0      .1       0   246.5    .045       0   287.4      .1       0
Bank Sta=246.5,287.4
XS Rating Curve= 0 ,0
Exp/Cntr(USF)=0,0
Exp/Cntr=0.3,0.1

Type RM Length L Ch R = 1 ,77599   ,125.3,121.4,117.9
XS GIS Cut Line= 3
2218910.91990602 642921.321220422218880.24465835 643094.52640357
2218843.04364157643321.140312407
#Sta/Elev= 30
       0 2661.89       8 2660.65    24.2 2656.04    38.7 2653.14    40.5  2652.6
    48.6  2648.3    60.8 2646.89    64.9 2645.27      77 2634.79    81.1 2632.24
    84.6 2630.99    89.2 2630.35    97.3 2630.07   109.5 2630.78   125.8 2632.17
   133.9 2631.76   154.1 2631.66   174.5  2632.2   185.2 2631.68   320.5 2631.75
   328.6 2632.27   340.7 2633.89   344.8 2633.11   348.9 2633.15   352.9  2633.6
     361 2635.31   369.1 2638.39   385.3 2643.08   393.4 2644.78   405.5  2646.7
#Mann= 3 ,-1,0
       0      .1       0    84.6    .045       0   109.5      .1       0
Bank Sta=84.6,109.5
XS Rating Curve= 0 ,0
Exp/Cntr(USF)=0,0
Exp/Cntr=0.3,0.1

Type RM Length L Ch R = 1 ,77477   ,188.9,189,188.4
XS GIS Cut Line= 3
2218759.20896688 642902.735504122218782.69076029643084.607135907
2218718.67990964 643314.13404047
#Sta/Elev= 30
       0 2655.49     6.5 2654.55    26.7 2650.42      63 2644.12      71 2643.02
    75.1 2641.47    95.2 2639.92    99.3 2638.73   110.2 2632.03   113.12630.782
   115.4 2629.93   119.4 2629.16   127.5 2628.75   135.8 2630.56   143.6 2631.23
   159.8 2631.47   171.9 2632.25   192.4 2632.34   200.6 2631.81   221.6 2631.72
   322.3 2631.95   325.5 2632.33   337.6 2637.77   341.7 2639.25   345.9 2640.19
   354.2 2641.18     371 2642.23   395.8 2644.55   416.5  2646.9   421.7 2646.98
#Mann= 3 ,-1,0
       0      .1       0   113.1    .045       0   135.8      .1       0
Bank Sta=113.1,135.8
XS Rating Curve= 0 ,0
Exp/Cntr(USF)=0,0
Exp/Cntr=0.3,0.1

Type RM Length L Ch R = 1 ,77288   ,280.4,285,281.1
XS GIS Cut Line= 3
2218640.60013798642886.9925515132218614.49102147643045.655644193
 2218574.3231499643320.805564411
#Sta/Elev= 30
       0 2653.84    34.6 2649.39    42.8 2646.74    64.9 2644.31    75.4 2641.09
    83.3 2636.82    91.4 2631.12    96.3 2628.91   131.1  2628.3   141.5 2630.02
   152.2 2630.07     173 2628.09   192.7 2628.08   198.62626.418   200.7 2625.53
   204.7 2625.31   211.8 2626.54   216.9 2628.08     221 2628.36   249.2 2627.81
   269.5  2625.7   278.8 2626.81   293.7 2626.49   297.8 2626.96   309.9  2633.1
   326.1  2636.4   350.3 2639.42   386.7 2642.63   398.9 2642.57   438.9 2648.09
#Mann= 5 ,-1,0
       0      .1       0      90     .12       0   190.8      .1       0
   198.6    .045       0   211.8      .1       0
Bank Sta=198.6,211.8
XS Rating Curve= 0 ,0
Exp/Cntr(USF)=0,0
Exp/Cntr=0.3,0.1

Type RM Length L Ch R = 1 ,77003   ,242.9,241.6,236.8
XS GIS Cut Line= 3
2218504.29660259642879.9148609672218477.14702662643068.260113916
2218440.54405366643339.122113844
#Sta/Elev= 30
       0  2658.8     9.4 2653.86    17.4 2647.25    21.5 2645.36    37.6 2644.71
    48.6 2638.65    61.9 2634.49    65.9 2632.89      74 2628.12    78.1 2627.12
     139  2626.1     171 2628.74   199.3  2628.6   215.4 2627.16   234.6 2628.77
   239.7 2628.13   247.7 2625.25   254.32624.117   263.9 2622.91   271.9 2623.22
   275.92624.118   280.9 2625.83   292.1 2632.96   300.2  2635.5   323.5 2637.29
   336.5 2637.16   398.2 2639.85   409.2 2640.73   449.5 2646.29   463.6 2645.67
#Mann= 5 ,-1,0
       0      .1       0     100     .12       0  200.29      .1       0
   254.3    .045       0   275.9      .1       0
Bank Sta=254.3,275.9
XS Rating Curve= 0 ,0
Exp/Cntr(USF)=0,0
Exp/Cntr=0.3,0.1

Type RM Length L Ch R = 1 ,76762   ,107.5,106.5,102.5
XS GIS Cut Line= 5
2218223.73675947642926.9990522342218251.48766945642995.308984497
2218287.77732097643081.7637425172218349.88846322643167.413586244
2218402.32881053643341.361894657
#Sta/Elev= 30
       0 2632.29    11.2 2630.39    36.9  2631.4    88.8 2628.86      94 2627.95
    97.1 2626.27   101.12623.329   101.8 2622.88   106.1 2622.57   116.8 2623.04
   127.8 2623.91   145.2 2624.45   158.2 2626.47   162.5 2626.74   176.7 2624.74
     239 2625.02   245.8 2625.54   255.7 2625.29   260.7 2626.68   267.6 2629.66
   273.3 2631.46   283.5 2632.53   312.7 2633.68   354.5  2632.7   375.4 2636.69
   408.8 2640.37   417.8    2642   429.7 2642.73   442.3 2645.38     455    2646
#Mann= 5 ,-1,0
       0      .1       0   101.1    .045       0   116.8      .1       0
   267.6     .12       0   283.5      .1       0
Bank Sta=101.1,116.8
XS Rating Curve= 0 ,0
Exp/Cntr(USF)=0,0
Exp/Cntr=0.3,0.1

Type RM Length L Ch R = 1 ,76655   ,154.4,158.3,156.5
XS GIS Cut Line= 3
 2218076.7069555642968.391156819 2218316.2078897  643241.3318441
2218328.27190164643395.895546245
#Sta/Elev= 30
       0 2651.59    47.7 2637.56    65.9 2628.74      71 2627.09    85.2 2626.29
   102.3 2626.28   134.1 2623.36   171.3 2621.36   181.1 2620.47   188.1 2621.47
   192.9 2623.29   203.3 2623.75   232.6 2622.97   247.8 2623.39   286.5  2621.6
   299.1 2621.72   304.4 2623.14   309.1 2625.52     315 2627.52   332.7  2629.9
     346 2632.55   362.9 2634.43     387 2635.79   423.2 2636.63   443.2 2638.11
   459.3 2640.88   467.3 2642.85   483.3 2644.39   487.3 2645.74   518.2 2652.77
#Mann= 7 ,-1,0
       0      .1       0      10     .12       0     110      .1       0
   171.3    .045       0   188.1      .1       0     270     .12       0
  393.12      .1       0
Bank Sta=171.3,188.1
XS Rating Curve= 0 ,0
Exp/Cntr(USF)=0,0
Exp/Cntr=0.3,0.1

Type RM Length L Ch R = 1 ,76497   ,247.2,252.3,246.4
XS GIS Cut Line= 4
2217968.00953253 643038.282912872217983.49531436643058.480750143
2218227.27111429643378.3907338422218251.02237675643428.789362294
#Sta/Elev= 30
       0 2663.61    27.9 2658.92    43.9 2653.59      59 2649.93    69.1 2645.38
    84.9  2634.8   104.9  2624.3   109.3  2622.5     122 2619.88   134.5 2618.85
   164.6 2621.22   178.4 2621.32   207.7 2619.67   214.9 2621.14   219.32619.903
     230  2618.6   237.8  2620.2   244.8 2622.07   275.3 2620.39     284 2618.93
     319 2621.27   335.6 2619.75   353.1 2619.95   358.9 2621.66   380.9 2633.69
     406 2636.16   427.7  2640.1   439.6 2640.92   448.4 2644.81   483.4 2655.11
#Mann= 3 ,-1,0
       0      .1       0   219.3    .045       0   237.8      .1       0
Bank Sta=219.3,237.8
XS Rating Curve= 0 ,0
Exp/Cntr(USF)=0,0
Exp/Cntr=0.3,0.1

Type RM Length L Ch R = 1 ,76245   ,253.5,255.9,255.7
XS GIS Cut Line= 5
2217803.51379331643122.5265245372217855.39059943643179.252596957
 2217967.3956967643303.7027050322218009.85514534643353.482748262
2218027.47200953643553.850969175
#Sta/Elev= 30
       0 2674.16     5.2 2673.47    14.4 2668.66    22.2 2666.25    74.1 2653.69
    90.1 2648.62   113.9 2636.31   133.3 2630.24   143.8 2625.79   155.2 2616.33
   165.6 2615.32   174.52616.321   191.7 2617.22   203.2 2619.04   209.6 2618.32
   251.6 2619.24   262.9 2617.76   274.3 2619.56   317.5 2619.19   325.5 2617.76
   333.5 2617.96   345.6 2616.56   349.6 2617.73   365.6 2628.68   393.7 2637.28
   413.8  2639.1   417.8 2641.28     426 2643.72   474.1 2652.83   510.9 2658.47
#Mann= 3 ,-1,0
       0      .1       0   155.2    .045       0   174.5      .1       0
Bank Sta=155.2,174.5
XS Rating Curve= 0 ,0
Exp/Cntr(USF)=0,0
Exp/Cntr=0.3,0.1

Type RM Length L Ch R = 1 ,75989   ,221.5,221.1,219.9
XS GIS Cut Line= 2
2217610.46488122643192.9460654362217859.00358652643557.168240848
#Sta/Elev= 30
       0 2674.46    14.8 2669.93    19.7 2667.46    24.3 2665.94    38.8 2665.32
    43.9 2664.42    58.4 2658.71    76.2 2653.89    95.3 2650.27   111.7 2648.32
   123.7 2645.75   135.9  2644.1     154 2639.31   174.1  2631.6   179.5 2628.34
   189.1 2620.71   203.1 2614.06   208.6 2612.82   213.4 2612.71   222.52614.056
   227.9 2614.57   269.1 2614.72   281.2  2616.7   306.5 2618.76   322.4 2621.36
   339.3 2625.68   369.8 2631.47   418.8 2639.82   428.8 2640.98   440.9 2641.19
#Mann= 3 ,-1,0
       0      .1       0   203.1    .045       0   222.5      .1       0
Bank Sta=203.1,222.5
XS Rating Curve= 0 ,0
Exp/Cntr(USF)=0,0
Exp/Cntr=0.3,0.1

Type RM Length L Ch R = 1 ,75768   ,243,244.2,242
XS GIS Cut Line= 2
2217434.34902315643344.2334566752217707.77323118643693.425818744
#Sta/Elev= 30
       0 2652.85     4.8 2651.77    15.9 2646.24    35.4 2640.85    41.9 2639.78
    72.3 2637.14    82.5 2634.87      96 2632.93   107.9 2630.25   126.2 2627.22
   147.3 2621.96   163.8 2615.76   168.9 2614.43   178.6 2613.72     190 2614.35
   204.1 2613.12     2092611.767   217.1 2610.95   227.1 2611.76     243 2612.98
   281.2 2611.38   298.3 2611.57   306.8 2613.57   311.1 2615.81   320.9  2622.3
   326.3 2623.82   397.5 2633.53     418 2636.89   431.2 2640.58   443.5 2641.51
#Mann= 3 ,-1,0
       0      .1       0     209    .045       0   227.1      .1       0
Bank Sta=209,227.1
XS Rating Curve= 0 ,0
Exp/Cntr(USF)=0,0
Exp/Cntr=0.3,0.1

Type RM Length L Ch R = 1 ,75523   ,201.4,197,190.3
XS GIS Cut Line= 2
2217234.72977961643467.3848966972217557.51966701643893.782552013
#Sta/Elev= 30
       0 2654.95    62.3 2642.48    95.2 2635.25   141.6 2631.71   157.8 2629.46
   179.3  2624.9   185.1 2622.36   201.2 2611.27   206.52608.728     213 2607.68
     223 2608.04     228 2609.24   234.3 2611.04   258.1 2612.79   278.2 2612.55
   287.4 2613.03   298.2 2609.05   303.3 2608.27   320.5 2608.94   339.2 2611.22
   358.4 2611.51   378.5 2617.59     400 2621.23   416.3 2625.33     453 2633.26
   473.8 2636.98   487.7 2640.54   499.4  2642.3   510.6  2645.6   534.8 2654.11
#Mann= 3 ,-1,0
       0      .1       0   206.5    .045       0     228      .1       0
Bank Sta=206.5,228
XS Rating Curve= 0 ,0
Exp/Cntr(USF)=0,0
Exp/Cntr=0.3,0.1

Type RM Length L Ch R = 1 ,75326   ,122.6,128.9,134.8
XS GIS Cut Line= 4
2217097.92681203643680.1738772712217233.49337856643782.300690724
2217301.27666183 643808.510226922217506.43406584643904.310600602
#Sta/Elev= 30
       0 2643.21    10.9 2640.31    26.6 2634.49    33.7 2632.83      48 2628.18
    70.9 2625.45     108 2618.25   121.3 2613.98   134.6 2608.33   145.1 2607.29
   176.9 2608.58   189.8 2608.16     194 2606.92   198.3 2605.63   202.6 2605.47
   211.3 2606.45   229.7 2609.68   248.1 2610.99   275.2 2610.67   294.2  2607.2
   342.7 2609.01   359.4 2608.72   365.5 2611.67     378  2621.7   385.8 2625.28
   401.6 2627.51   417.8 2630.83   442.5 2636.35   457.5 2640.74   468.8 2643.18
#Mann= 3 ,-1,0
       0      .1       0     194    .045       0   211.3      .1       0
Bank Sta=194,211.3
XS Rating Curve= 0 ,0
Exp/Cntr(USF)=0,0
Exp/Cntr=0.3,0.1

Type RM Length L Ch R = 1 ,75198   ,264.9,269,268.4
XS GIS Cut Line= 5
2217046.24328176643723.310412701 2217132.6077868643803.850336588
2217163.82756054643854.0154430972217193.03247122643966.874694909
2217248.37303246644116.670362146
#Sta/Elev= 30
       0 2645.03    13.6 2639.57    20.3 2637.56    49.7  2631.5    84.7 2625.89
    90.2 2624.51   108.3 2614.87   124.5 2606.98   130.4  2606.4     140 2607.11
   143.2  2606.8   147.9  2605.3   152.6 2604.36   157.3 2604.14   162.7  2605.1
   166.8    2607   176.2 2607.48   201.1 2605.51   229.3 2604.56   238.3 2605.47
   246.6 2605.48   263.1 2603.03   294.9 2606.54   321.8 2608.54   347.4 2614.05
   366.5 2616.63   381.5 2617.68   393.8 2619.63   436.9 2628.78   453.4 2631.26
#Mann= 3 ,-1,0
       0      .1       0   147.9    .045       0   162.7      .1       0
Bank Sta=147.9,162.7
XS Rating Curve= 0 ,0
Exp/Cntr(USF)=0,0
Exp/Cntr=0.3,0.1

Type RM Length L Ch R = 1 ,74929   ,204.5,203.7,200.2
XS GIS Cut Line= 2
2216869.38798649643818.4476445772217066.11371325644235.498356342
#Sta/Elev= 30
       0 2663.02    16.2 2655.22    31.2 2651.03    47.2 2644.94    62.8 2641.12
    73.3 2637.28    82.3 2636.29   109.3 2625.58   124.4 2620.48     149 2607.71
   157.8 2604.24   166.4  2602.3   184.52601.176   193.2 2599.92     202 2600.35
     2042601.181   210.9 2604.55   215.3 2604.71   224.2 2602.53   228.6 2603.25
   241.8 2610.52   255.1 2612.94   269.1 2613.98   299.3 2620.65   316.7 2623.58
   337.7 2629.08   388.8 2638.64   409.9 2643.54   440.9 2653.44   461.1 2657.78
#Mann= 3 ,-1,0
       0      .1       0   184.5    .045       0     204      .1       0
Bank Sta=184.5,204
XS Rating Curve= 0 ,0
Exp/Cntr(USF)=0,0
Exp/Cntr=0.3,0.1

Type RM Length L Ch R = 1 ,74725   ,239,239.3,236.3
XS GIS Cut Line= 2
2216639.84817476643880.5859643882216925.44174158644304.457429073
#Sta/Elev= 30
       0 2677.86      20 2671.72    35.2 2665.92    53.8 2659.99      65 2654.21
    68.2 2653.34    78.5 2652.66   106.8 2642.82   116.5 2640.48   136.1 2633.83
   150.9 2630.88   165.2 2624.47   179.3 2619.15     208 2609.96   228.62599.989
   236.8 2598.97   257.32599.995   265.5 2601.31   279.8 2605.16   294.9 2606.77
     319 2612.93   343.2 2619.69   366.6 2627.28   386.6 2632.06     401 2636.39
   410.7 2637.59   449.3 2646.27   458.7 2649.87   492.7 2660.12   511.1 2666.78
#Mann= 3 ,-1,0
       0      .1       0   228.6    .045       0   257.3      .1       0
Bank Sta=228.6,257.3
XS Rating Curve= 0 ,0
Exp/Cntr(USF)=0,0
Exp/Cntr=0.3,0.1

Type RM Length L Ch R = 1 ,74486   ,280.5,280,279.1
XS GIS Cut Line= 2
2216452.88904811644052.1883186582216782.79006926644464.017751488
#Sta/Elev= 30
       0    2651    11.7 2649.89      40 2645.65      50 2643.74      60 2640.89
      82 2632.77    98.6 2625.96   124.3 2614.44   152.4 2604.37   170.9 2601.84
   185.2 2601.39   193.7 2599.94     210 2599.55   218.62597.256   227.8 2596.45
   239.52597.252   242.2 2597.64   252.4 2600.82   267.6 2603.76   281.9 2608.19
   301.8 2612.93   313.9 2614.85   330.3 2619.96   367.3 2628.89   421.3 2644.47
   444.1 2650.29     464 2654.62   485.1 2657.71   513.8 2664.07   527.7  2667.8
#Mann= 3 ,-1,0
       0      .1       0   218.6    .045       0   239.5      .1       0
Bank Sta=218.6,239.5
XS Rating Curve= 0 ,0
Exp/Cntr(USF)=0,0
Exp/Cntr=0.3,0.1

Type RM Length L Ch R = 1 ,74206   ,221.6,223.7,226.2
XS GIS Cut Line= 3
2216078.10535354644249.0845879832216312.24434843644334.186296713
2216567.97208368644607.923000791
#Sta/Elev= 30
       0 2620.64    57.5 2612.78    70.3 2608.81    78.8 2607.46    95.8 2607.46
   112.9 2609.36   117.2 2609.11   121.4 2608.04   134.1 2602.04   146.9 2598.57
   155.4 2598.64   168.2    2601   185.2 2601.51   236.3 2599.23   249.1 2599.61
   302.1 2598.25   313.5  2597.5   331.1 2593.72   342.8 2594.97   354.5 2594.89
     3642593.106   378.5 2591.75     3902593.115   406.5 2601.55   429.5  2604.5
   454.1 2609.54   500.2 2624.38   570.7 2638.85     605 2649.87   623.7 2654.92
#Mann= 5 ,-1,0
       0      .1       0     220     .06       0  349.13      .1       0
     364    .045       0     390      .1       0
Bank Sta=364,390
XS Rating Curve= 0 ,0
Exp/Cntr(USF)=0,0
Exp/Cntr=0.3,0.1

Type RM Length L Ch R = 1 ,73982   ,294.3,290,283.1
XS GIS Cut Line= 6
 2215971.1209116644400.3976857612216165.60775178644472.804054181
2216203.16240204644531.4420168682216239.39934528644592.056540095
2216264.68047923644641.7888839782216342.83934687 644719.21526817
#Sta/Elev= 30
       0 2628.44    13.7 2625.53    36.6 2617.43    48.1 2614.59    60.5 2612.22
    79.2 2611.15   107.8 2606.06   116.5  2605.6   137.7 2606.55   151.3 2605.21
   163.3 2600.97   197.7 2600.73   212.3 2598.27   219.7 2594.93   224.1 2594.19
   244.4 2593.49   269.7 2594.42   279.2 2593.09   299.6 2592.69   305.12590.936
   311.8 2589.69   321.22590.973   325.8 2593.57   330.4 2594.56   352.2 2594.34
     376 2596.28   393.9 2598.88   405.6 2601.47   419.8 2602.72   513.6 2617.07
#Mann= 5 ,-1,0
       0      .1       0     140     .06       0  297.16      .1       0
   305.1    .045       0   321.2      .1       0
Bank Sta=305.1,321.2
XS Rating Curve= 0 ,0
Exp/Cntr(USF)=0,0
Exp/Cntr=0.3,0.1

Type RM Length L Ch R = 1 ,73692   ,272.5,271,258.2
XS GIS Cut Line= 4
2215821.82274198644749.5214703062215969.13841094644735.061036543
 2216160.7391583644822.7274162332216299.85883571644811.483019732
#Sta/Elev= 30
       0 2645.21    24.4 2637.34    54.6 2629.23    78.7 2620.61    98.8 2615.74
   102.8 2614.24   114.9 2604.55   172.3 2600.99   182.3 2595.92   191.1 2592.59
   212.9 2588.77   226.1 2587.66   234.9 2589.11   243.7  2590.4   261.3 2590.48
   274.5 2586.86   278.9 2586.72   287.7  2587.5   296.5 2590.19   317.9 2588.84
   331.7 2586.82   349.3 2588.12     355 2589.97   362.2  2590.6   374.2  2587.6
   378.2  2587.5   421.9 2596.24   438.4 2598.42   478.7 2610.64   498.3 2614.91
#Mann= 5 ,-1,0
       0      .1       0  168.02     .06       0   212.9    .045       0
   234.9     .06       0  278.02      .1       0
Bank Sta=212.9,234.9
XS Rating Curve= 0 ,0
Exp/Cntr(USF)=0,0
Exp/Cntr=0.3,0.1

Type RM Length L Ch R = 1 ,73421   ,198.2,198.3,197.1
XS GIS Cut Line= 3
2215916.58824168644976.5425422342216079.52317952644928.741614585
2216310.46930686644908.621555696
#Sta/Elev= 30
       0  2616.6     3.7 2615.12    28.7 2608.07    41.3  2602.5    57.2 2602.37
    62.1  2601.5    66.3 2598.76    74.6  2591.3    78.8 2588.83    86.2 2586.25
    91.3  2585.9   103.8 2586.74   116.3 2589.29   131.3 2589.17   144.2 2590.09
   182.5 2590.24   203.2 2589.92   210.6 2590.34   226.7 2588.82   238.7 2590.48
   267.32587.233   278.9 2586.06   284.12587.228   302.9 2592.81     311 2594.09
     327 2598.39   335.1 2599.96   351.1  2605.6   359.2 2607.02   401.6  2620.6
#Mann= 5 ,-1,0
       0      .1       0   131.3     .06       0   182.5      .1       0
   267.3    .045       0   284.1      .1       0
Bank Sta=267.3,284.1
XS Rating Curve= 0 ,0
Exp/Cntr(USF)=0,0
Exp/Cntr=0.3,0.1

Type RM Length L Ch R = 1 ,73223   ,217.9,212.5,207.5
XS GIS Cut Line= 4
2215951.81758616645175.3498514472216126.41376719 645116.71188876
2216209.42930987645110.1233536272216373.79202269645091.033773505
#Sta/Elev= 30
       0 2625.74    63.7 2603.72    80.5 2599.69    84.8 2598.91    96.8 2599.31
   110.1    2599     127 2595.92   131.2 2594.98   134.7 2593.59   148.1 2586.83
   156.8 2585.35   166.2 2583.05   170.1 2582.85   181.8 2584.13     194 2584.07
   212.42582.711     218 2582.35   235.52582.525   243.3 2583.16   258.2 2586.23
   267.2 2586.55   282.3 2586.17   306.5 2590.85   338.7 2600.31   366.9 2609.36
   378.9 2612.17   399.1 2619.79   415.1 2624.08   427.3  2626.7   432.9 2628.64
#Mann= 5 ,-1,0
       0      .1       0     140     .06       0   212.4    .045       0
   235.5     .06       0  244.18      .1       0
Bank Sta=212.4,235.5
XS Rating Curve= 0 ,0
Exp/Cntr(USF)=0,0
Exp/Cntr=0.3,0.1

Type RM Length L Ch R = 1 ,73010   ,259,264.1,266.1
XS GIS Cut Line= 4
2215966.11198455645357.8081817952216198.58815655645325.001151203
2216297.09986156 645265.351861932216440.95518201645260.189754421
#Sta/Elev= 30
       0 2649.37     6.1 2649.29    34.4 2643.31    62.7 2635.11    82.9 2626.72
      99 2624.61   111.2 2620.27   127.3 2616.65   139.4 2612.34   152.2 2609.17
   183.9 2599.32     190 2596.69     196  2592.5     200 2591.14   220.2 2591.98
   228.3 2590.66   236.6 2586.87   241.3 2585.62     262 2583.97   294.1 2584.33
   309.52580.197   316.1 2579.54   326.32580.198   330.2 2580.62   344.2 2584.34
   356.9 2593.65     365 2598.15   449.1 2626.91   461.1 2633.96   493.9 2642.61
#Mann= 5 ,-1,0
       0      .1       0     220     .06       0   309.5    .045       0
   326.3     .06       0  334.78      .1       0
Bank Sta=309.5,326.3
XS Rating Curve= 0 ,0
Exp/Cntr(USF)=0,0
Exp/Cntr=0.3,0.1

Type RM Length L Ch R = 1 ,72746   ,240.1,241.9,244.7
XS GIS Cut Line= 4
2216003.31930471645555.4618666962216132.96813908645545.742403722
2216418.47132819645518.0868241492216607.17033436645566.306034036
#Sta/Elev= 30
       0 2638.51    20.9  2638.1      49 2634.78      61 2635.28    76.5  2627.7
   133.2    2613   145.3 2610.87   169.4 2600.68   181.5 2592.03   205.6 2590.28
   217.7 2583.93   237.7 2578.22   245.8 2577.58     258 2579.77   273.9 2580.51
   293.52577.091   310.1 2576.11   317.72577.084   338.2 2580.07   358.3 2584.45
   386.4 2592.69   418.6  2599.6   435.1 2601.47   443.8 2600.72   451.6 2598.56
   472.3 2598.52   499.7 2603.48   521.8 2605.84   539.2 2609.26   611.6 2629.32
#Mann= 3 ,-1,0
       0      .1       0   293.5    .045       0   317.7      .1       0
Bank Sta=293.5,317.7
XS Rating Curve= 0 ,0
Exp/Cntr(USF)=0,0
Exp/Cntr=0.3,0.1

Type RM Length L Ch R = 1 ,72504   ,167.7,181.5,194.2
XS GIS Cut Line= 4
2216055.80062479645670.192398587 2216270.2277814645758.175213476
2216480.86874042645766.8922201552216537.00961905645768.770587838
#Sta/Elev= 30
       0 2610.32    17.7 2608.47    52.3 2603.05    86.9 2592.33    91.5 2590.12
    99.8 2584.02   103.7 2582.55   125.8 2583.05   137.5 2578.95   158.9    2573
     162 2572.68     169  2573.1     182 2575.26     195 2575.02   253.7 2577.92
   277.8 2577.26   285.8 2574.86     2912574.663   305.8 2573.28   325.92574.058
   333.8  2577.1   341.8 2583.88   349.8 2588.34   353.8 2589.85   417.2 2612.38
   433.9 2616.75   449.9 2625.64   461.9 2629.25   485.1 2634.51   498.8 2639.22
#Mann= 5 ,-1,0
       0      .1       0     140     .06       0  241.78      .1       0
     291    .045       0   325.9      .1       0
Bank Sta=291,325.9
XS Rating Curve= 0 ,0
Exp/Cntr(USF)=0,0
Exp/Cntr=0.3,0.1

Type RM Length L Ch R = 1 ,72323   ,198.7,198.8,194.8
XS GIS Cut Line= 3
2216023.54429403645731.1573194532216219.92055502645838.271643625
2216322.57178235 646041.34254987
#Sta/Elev= 30
       0 2599.13    28.1 2597.35    46.2 2594.21    78.6 2584.38    87.5 2580.26
    91.8 2579.07   119.2 2580.54   122.8 2579.69   131.7 2576.27   146.2 2573.13
     173 2570.45   184.7 2572.99   196.3 2574.84   201.2 2575.09     226  2574.8
   235.9 2573.79   249.9 2574.17   267.3 2572.61   285.2 2573.24   291.62572.086
   303.4 2570.63   309.52571.428   312.4 2572.81   321.3  2579.4   330.2  2589.7
   333.2 2591.03   357.3 2596.14   374.9 2602.03   389.8 2605.28   451.2 2624.33
#Mann= 5 ,-1,0
       0      .1       0      70     .06       0     210      .1       0
   291.6    .045       0   309.5      .1       0
Bank Sta=291.6,309.5
XS Rating Curve= 0 ,0
Exp/Cntr(USF)=0,0
Exp/Cntr=0.3,0.1

Type RM Length L Ch R = 1 ,72124   ,156.8,155.8,154.4
XS GIS Cut Line= 4
2215960.37446488645811.1140341572216073.79656046645933.046882533
2216124.40807863646000.8301657992216199.37832168646072.929225213
#Sta/Elev= 30
       0 2591.85    19.2 2586.68    60.8  2578.8    69.2 2575.68    80.6 2575.99
    97.5 2575.37   101.2 2574.57   106.6 2571.87   111.3 2570.31     123 2569.06
   144.9 2568.33   161.2 2570.05   176.7 2570.22   181.7 2569.08   189.12566.004
   191.7 2565.26   201.6 2564.53   205.5 2564.81   209.92566.012   216.9 2568.99
   231.6 2569.76   236.6 2571.45   246.6 2579.06   250.7  2581.5   267.4 2587.73
   276.7 2589.57   299.3 2596.42   322.9 2604.97     334 2606.64   355.1 2612.51
#Mann= 5 ,-1,0
       0      .1       0      30     .06       0     160      .1       0
   189.1    .045       0   209.9      .1       0
Bank Sta=189.1,209.9
XS Rating Curve= 0 ,0
Exp/Cntr(USF)=0,0
Exp/Cntr=0.3,0.1

Type RM Length L Ch R = 1 ,71968   ,205.9,197.5,190.8
XS GIS Cut Line= 3
2215806.82548815645856.122947632 2215999.8544265646078.162015449
2216169.45210644646129.487629115
#Sta/Elev= 30
       0  2607.9      12 2604.75    54.4 2590.71    75.6 2587.02    86.8 2584.32
   103.8    2577   139.2 2575.66   149.1 2569.74   154.5  2567.8   178.9 2562.98
   186.9 2563.24   197.3 2565.56   200.2 2565.69   203.3 2565.57   209.92563.948
   217.2 2562.48   225.7 2562.27   233.42563.229     252 2565.18   270.3 2565.63
   282.5 2569.22   288.6 2569.96   300.1 2570.18     328 2574.29   357.2 2580.83
   386.5 2586.54     399 2590.48   411.6 2592.31   428.9 2596.92   471.4 2606.19
#Mann= 4 ,-1,0
       0      .1       0     120     .06       0   209.9    .045       0
   233.4      .1       0
Bank Sta=209.9,233.4
XS Rating Curve= 0 ,0
Exp/Cntr(USF)=0,0
Exp/Cntr=0.3,0.1

Type RM Length L Ch R = 1 ,71771   ,175.4,162.6,153.3
XS GIS Cut Line= 3
2215758.33203685646168.8835330712215914.91120971646201.063915223
2216094.54498471646151.112277256
#Sta/Elev= 30
       0 2577.29    22.3 2574.01    26.4 2573.05      38 2569.48    46.8 2564.98
      55 2561.75    59.1 2560.65    75.4 2559.78    82.42557.817    93.3 2556.69
    99.9 2556.87   105.52558.122   108.1 2559.01   112.1 2559.56   123.8 2559.21
   132.6 2559.89   148.9 2559.96   193.3 2557.78   202.7 2559.19   206.8  2559.4
   219.1 2558.07   223.4 2558.37     229 2559.51     240 2562.81   244.2 2563.45
     294 2569.03   306.5  2571.9   318.9 2575.49   331.4 2577.42   346.3 2582.46
#Mann= 5 ,-1,0
       0      .1       0      30     .06       0    82.4    .045       0
   105.5     .06       0  339.85      .1       0
Bank Sta=82.4,105.5
XS Rating Curve= 0 ,0
Exp/Cntr(USF)=0,0
Exp/Cntr=0.3,0.1

Type RM Length L Ch R = 1 ,71608   ,116.9,118.1,117.2
XS GIS Cut Line= 4
2215796.46669782646393.9426956072215902.60799882646352.434924266
2216041.36254873646206.5647564122216118.44840979646170.986666692
#Sta/Elev= 30
       0  2578.6    13.1 2578.29    24.1 2576.61    55.5 2567.75    68.3 2561.91
      77 2556.48    81.3 2554.82    85.6 2554.18    94.2 2554.57    98.5 2553.96
     122  2555.9   131.5 2553.78     140 2553.52   145.7 2554.04   150.32553.134
   154.2 2552.44   159.8 2552.34   167.82552.636   179.2 2554.51   209.1  2552.8
   219.2 2552.81   233.4  2556.3   264.5 2556.67   292.8 2562.67   306.9 2564.03
   324.5 2564.79   344.8 2568.12   357.6  2572.1   366.7 2573.88   400.2 2585.46
#Mann= 5 ,-1,0
       0      .1       0   150.3    .045       0   167.8      .1       0
  233.97     .06       0  365.29      .1       0
Bank Sta=150.3,167.8
XS Rating Curve= 0 ,0
Exp/Cntr(USF)=0,0
Exp/Cntr=0.3,0.1

Type RM Length L Ch R = 1 ,71490   ,206.1,207.4,207
XS GIS Cut Line= 4
2215808.11291024646539.2865991392215965.98406723646464.022772044
 2216149.4508206646214.5802896272216169.58601169646189.589433955
#Sta/Elev= 30
       0 2592.79    53.2 2578.78   133.7 2563.42   148.7 2556.81   155.2 2554.97
   163.7  2554.4   183.4 2554.88   188.4 2554.16   198.5 2550.52   201.4 2550.26
   218.1 2551.98     233 2552.39   238.6 2551.92   247.9 2549.22   266.4 2549.66
   278.6 2550.76   282.7 2550.52   290.42548.608   306.9 2547.44     3152548.598
   327.3 2552.77   367.3 2551.11     387 2558.94   391.9 2560.27   408.1 2562.18
   431.7  2567.8   461.7 2578.47   481.8  2584.5   491.5 2588.52   516.6 2595.57
#Mann= 5 ,-1,0
       0      .1       0   290.4    .045       0     315      .1       0
  354.89     .06       0  484.54      .1       0
Bank Sta=290.4,315
XS Rating Curve= 0 ,0
Exp/Cntr(USF)=0,0
Exp/Cntr=0.3,0.1

Type RM Length L Ch R = 1 ,71282   ,173.5,184.8,192.5
XS GIS Cut Line= 4
2215942.64231398 646607.16286546 2216147.4121254646560.383766004
2216279.36358349646385.954783734 2216315.5146679646332.631934231
#Sta/Elev= 30
       0 2560.61    22.1 2555.67      59 2549.11    67.2 2548.32   129.9 2548.01
   141.1 2549.09   145.2 2548.83   156.6    2545   161.6 2544.53   170.6 2544.74
   186.6 2547.98   202.6 2547.63   215.7 2545.68   224.1 2545.38   259.2 2545.51
   274.3 2546.66   287.22543.095   297.5 2542.11   306.72543.089   315.7 2546.54
   324.2 2551.05   341.4 2555.77   361.4 2558.61   384.6 2565.73   409.7 2574.74
   434.5 2580.57     449  2585.4   458.7 2586.75     478 2592.04   493.2 2594.19
#Mann= 5 ,-1,0
       0      .1       0  270.05     .06       0   287.2    .045       0
   306.7     .06       0  390.05      .1       0
Bank Sta=287.2,306.7
XS Rating Curve= 0 ,0
Exp/Cntr(USF)=0,0
Exp/Cntr=0.3,0.1

Type RM Length L Ch R = 1 ,71098   ,156.3,157.2,157.1
XS GIS Cut Line= 3
2215996.91619635646652.297688793 2216327.2587594646663.504787055
2216407.30946127646668.307829167
#Sta/Elev= 30
       0 2549.03    27.3 2546.31    63.3 2546.06    91.3 2544.08   127.3 2544.51
   139.3 2541.06   151.3 2541.22   163.4 2544.05   183.4 2543.53   191.4 2542.25
   203.4 2543.89   207.4 2543.03   219.4 2536.84   223.72535.487   239.4 2534.58
     2452535.485   259.5 2543.18   271.4  2553.2     280 2557.94   291.4    2564
   315.4 2574.23   319.4 2575.48   336.8 2576.32   339.5 2577.22   351.5 2585.22
   371.5 2592.58   379.5  2594.1   387.6 2593.58   395.6 2596.09   410.7 2602.73
#Mann= 5 ,-1,0
       0      .1       0     190     .06       0   223.7    .045       0
     245     .06       0     280      .1       0
Bank Sta=223.7,245
XS Rating Curve= 0 ,0
Exp/Cntr(USF)=0,0
Exp/Cntr=0.3,0.1

Type RM Length L Ch R = 1 ,70940   ,131.9,132.1,131.9
XS GIS Cut Line= 2
2215941.72217629 646794.924251932216434.71491149646831.274866106
#Sta/Elev= 30
       0 2561.24    34.5 2555.11    82.7 2543.46   106.7 2539.03   118.8 2539.36
   134.8  2541.6   146.9 2539.96   178.9 2539.45     195 2538.03     203 2535.77
     207 2535.54     215 2535.77   223.1 2538.76   231.1 2539.21   259.2 2532.73
   267.82532.172   283.2 2531.51   294.52533.016   303.3 2536.87   315.3 2544.41
   331.3 2552.69   348.1  2554.9   355.4  2557.1   371.5 2564.02   395.5 2568.26
   415.9 2576.28   431.6 2580.78   443.7 2583.17   471.7 2586.37   494.3 2590.85
#Mann= 5 ,-1,0
       0      .1       0     240     .06       0   267.8    .045       0
   294.5     .06       0     440      .1       0
Bank Sta=267.8,294.5
XS Rating Curve= 0 ,0
Exp/Cntr(USF)=0,0
Exp/Cntr=0.3,0.1

Type RM Length L Ch R = 1 ,70808   ,210.1,213.3,209.2
XS GIS Cut Line= 3
2215904.22893912646928.3686701822215986.07139053646926.899878041
2216364.30211116646959.435854008
#Sta/Elev= 30
       0 2564.46      32 2556.74      48 2554.63      60 2551.22      76  2549.9
      84 2547.07     104 2542.61   152.2 2536.83   196.4 2534.92   216.5 2535.74
   228.5 2533.29   240.5 2532.68   252.6 2534.32   256.6 2535.24   264.6  2538.9
   268.6  2538.9   280.7 2532.87   288.7 2531.71   296.7 2532.79     304 2530.72
   316.8 2529.58   322.32530.741     353 2533.97     361  2537.4     373 2544.89
     377 2545.95   393.1 2547.22   401.1 2551.01   429.2 2558.21   461.5 2562.82
#Mann= 5 ,-1,0
       0      .1       0  181.86     .06       0     304    .045       0
   322.3     .06       0  381.86      .1       0
Bank Sta=304,322.3
XS Rating Curve= 0 ,0
Exp/Cntr(USF)=0,0
Exp/Cntr=0.3,0.1

Type RM Length L Ch R = 1 ,70595   ,131.3,134,136.7
XS GIS Cut Line= 4
2215930.88416911647098.7114523742216110.97079609647127.993830745
2216264.70328253647124.3335334482216374.51220143647058.448182114
#Sta/Elev= 30
       0 2549.23     9.4 2546.76    29.7 2540.39    41.8 2536.11    45.1 2535.72
    55.6 2535.48    66.1 2536.48    94.5 2533.81   118.8 2532.13   155.3 2530.77
   183.7 2529.09   211.7  2528.5   215.7 2528.05   221.6 2525.51   223.7 2524.55
   227.7 2524.09   231.7 2524.12   238.52525.516   243.7 2526.47   251.7 2526.99
   303.8 2527.66   319.7 2528.81   340.3 2529.49   387.7 2536.03   414.9 2534.66
   419.8 2535.53   431.4 2541.62   438.2 2543.85   452.2 2545.78   464.3 2546.36
#Mann= 5 ,-1,0
       0      .1       0      60     .06       0     160      .1       0
   221.6    .045       0   238.5      .1       0
Bank Sta=221.6,238.5
XS Rating Curve= 0 ,0
Exp/Cntr(USF)=0,0
Exp/Cntr=0.3,0.1

Type RM Length L Ch R = 1 ,70461   ,229.7,228.6,220.1
XS GIS Cut Line= 4
 2215865.5930012647250.9694137682216037.34035409647250.213802524
2216214.57194918647260.096605225 2216497.6669864647354.007934263
#Sta/Elev= 30
       0 2540.75    38.6 2538.84    42.6 2538.32    50.6 2535.16    54.6 2534.61
    74.6 2535.81    86.6 2535.45    98.6 2536.79   118.6 2532.98   138.6  2530.8
   226.8 2526.94   254.7 2527.27   270.7 2524.37   293.52524.177   306.8 2522.34
   313.9 2522.35   322.8  2522.7   329.22524.447   334.8 2526.62   338.8  2526.9
     372 2524.36   414.2  2525.2   422.6 2524.16     431 2521.46   435.2 2521.19
   468.9 2526.67   502.7 2529.63   604.5 2533.29   624.9 2535.03   647.5 2538.22
#Mann= 5 ,-1,0
       0     .05       0      20     .07       0     120      .1       0
   293.5    .045       0   329.2      .1       0
Bank Sta=293.5,329.2
XS Rating Curve= 0 ,0
Exp/Cntr(USF)=0,0
Exp/Cntr=0.3,0.1

Type RM Length L Ch R = 1 ,70232   ,212.4,229,242.2
XS GIS Cut Line= 4
2215918.07617905647445.2750020842216130.30045422647463.621541622
2216365.29154064647408.7170821772216467.77986494647386.755298399
#Sta/Elev= 30
       0 2529.78     6.1 2529.72    10.1 2528.69    22.2 2522.03    31.4 2520.23
    66.3 2522.92   130.6 2524.38   174.7 2522.19   223.3 2522.18   291.12518.264
   301.2 2516.46   313.5 2515.38   321.7 2515.79   329.62518.443   334.1 2519.74
   346.4 2521.25     371 2519.54   375.1 2519.58   383.4 2521.58   403.9 2521.31
     408 2521.85   416.2 2525.33   423.1  2527.3   432.7 2528.99   449.1 2529.08
   461.4 2530.27   481.8 2530.04     517 2531.01   547.2 2533.23   559.2 2535.27
#Mann= 4 ,-1,0
       0     .06       0     170      .1       0   291.1    .045       0
   329.6      .1       0
Bank Sta=291.1,329.6
XS Rating Curve= 0 ,0
Exp/Cntr(USF)=0,0
Exp/Cntr=0.3,0.1

Type RM Length L Ch R = 1 ,70003   ,332.6,331,325.4
XS GIS Cut Line= 3
2215892.21214266647555.3334794332216132.86274043647584.225642942
2216309.43548201647774.634308299
#Sta/Elev= 30
       0    2528      12 2524.01    28.2 2522.47      70 2515.33    92.6  2516.1
   112.8 2517.97   165.1 2519.29   185.3 2517.21   253.1 2518.67     260 2519.36
   276.5 2519.44   282.5 2520.22   288.4 2519.84   304.8 2514.78   309.52513.934
   320.1 2511.99   332.92513.929   341.4 2516.35   347.3 2519.07   358.2 2529.27
   361.4 2531.67   369.1 2535.97   375.6 2538.39   388.4 2542.22   400.2 2544.93
   412.4 2548.99   429.2 2551.75   437.9 2555.38   470.8 2564.25   502.1 2573.57
#Mann= 4 ,-1,0
       0     .06       0      90      .1       0   309.5    .045       0
   332.9      .1       0
Bank Sta=309.5,332.9
XS Rating Curve= 0 ,0
Exp/Cntr(USF)=0,0
Exp/Cntr=0.3,0.1

Type RM Length L Ch R = 1 ,69672   ,187.6,183.7,178.9
XS GIS Cut Line= 2
2215715.37412671647666.3815500222216069.19733636 647947.48563584
#Sta/Elev= 30
       0 2536.22     8.3 2535.98    13.9 2534.87    41.9 2526.65    55.9 2521.66
    77.7 2519.52   108.3  2512.5   113.4  2511.9   123.6 2511.32   144.1 2512.07
   159.4 2510.09   173.4 2512.16   197.4 2512.48   227.5 2511.65   241.1 2512.36
   244.5 2511.67   249.92509.246   255.9 2508.38     273 2508.27   284.72509.238
   292.9 2510.41   312.7 2510.87   317.8 2511.89   324.3 2514.75   333.1 2521.47
   349.9 2528.25   358.4 2530.28   369.8 2531.54   409.7 2545.98   451.9  2557.6
#Mann= 5 ,-1,0
       0      .1       0     220     .06       0   249.9    .045       0
   284.7     .06       0     340      .1       0
Bank Sta=249.9,284.7
XS Rating Curve= 0 ,0
Exp/Cntr(USF)=0,0
Exp/Cntr=0.3,0.1

Type RM Length L Ch R = 1 ,69489   ,248.4,252,255.8
XS GIS Cut Line= 4
2215539.45734567647876.3889937122215687.67679175647959.536487852
2215784.38094254647977.612030056 2216007.5588506648010.371397991
#Sta/Elev= 30
       0 2550.86    27.6 2544.93    51.3 2537.08    59.9 2532.06    74.2 2515.83
    80.4  2511.3    92.6 2504.96   106.9 2503.71   138.4 2507.01   186.7 2508.39
   207.1 2507.16   227.4  2508.8   247.8  2508.1   280.2 2511.16   285.4 2511.04
   292.4  2509.5   312.6 2510.01   324.42505.366   335.42505.443     349 2507.62
   381.3 2507.48   385.4  2508.5   389.4 2510.64   401.5  2521.3   409.6 2526.16
   413.7 2527.57   433.9 2531.85   447.6 2532.88   479.3 2539.39   493.9 2543.41
#Mann= 7 ,-1,0
       0      .1       0  278.33     .06       0   324.4    .045       0
   335.4     .06       0  368.33      .1       0  378.33     .06       0
  468.33      .1       0
Bank Sta=324.4,335.4
XS Rating Curve= 0 ,0
Exp/Cntr(USF)=0,0
Exp/Cntr=0.3,0.1

Type RM Length L Ch R = 1 ,69237   ,96.1,95.1,93.9
XS GIS Cut Line= 2
2215501.32036028648007.3373212082215965.28608437648387.778915768
#Sta/Elev= 30
       0 2537.81    29.6 2528.44    60.6 2507.47    70.9 2502.84   111.3  2501.7
   122.7 2503.22   148.5 2504.06   182.4 2502.56   205.4 2504.78   239.2 2505.28
   255.2 2502.18   267.7 2502.35     279 2504.09   292.7 2501.37   298.5 2501.26
   315.22502.308   324.4 2506.91   347.2  2525.1   356.2 2530.21     370 2535.03
     413  2552.5   443.9 2553.76   474.4 2546.12   506.4 2543.35   520.6 2536.85
   526.3 2536.25   534.8 2538.31   564.4  2541.2   577.9 2545.37     600 2554.33
#Mann= 8 ,-1,0
       0      .1       0     290     .06       0   292.7    .045       0
   315.2     .06       0     370      .1       0     450     .12       0
     500      .1       0     600     .12       0
Bank Sta=292.7,315.2
XS Rating Curve= 0 ,0
Exp/Cntr(USF)=0,0
Exp/Cntr=0.3,0.1

Type RM Length L Ch R = 1 ,69142   ,183.1,191.5,204.8
XS GIS Cut Line= 4
2215419.03424973648097.6517277462215548.60877403648178.178268266
2215697.94890372648285.0589493212215875.10729286648435.131138473
#Sta/Elev= 30
       0 2543.39    70.2 2522.41    78.9 2520.89    97.6 2508.74   114.4 2500.44
   168.7 2499.52   186.5 2501.67     206 2500.97   226.4 2503.84   253.9 2502.91
   265.2 2500.26   281.22500.143   289.1 2499.11   305.52500.393   329.3 2502.71
   346.4 2516.11   352.1 2519.23   375.8 2526.48   414.5 2541.41   431.5 2543.49
     444 2546.75   451.4 2547.21   459.7 2545.78   480.7 2538.43   491.1 2536.91
   506.9  2530.4   512.1 2529.47   533.7 2533.81   548.8 2539.94   568.4 2544.56
#Mann= 5 ,-1,0
       0      .1       0   281.2    .045       0   305.5      .1       0
  322.56     .06       0   456.2     .12       0
Bank Sta=281.2,305.5
XS Rating Curve= 0 ,0
Exp/Cntr(USF)=0,0
Exp/Cntr=0.3,0.1

Type RM Length L Ch R = 1 ,68950   ,61.7,62,62.1
XS GIS Cut Line= 5
 2215431.4729341648163.7548893652215577.07956055648344.939605536
 2215569.8321719648390.4004979572215561.26707623648448.379607131
2215580.37382812648599.915915202
#Sta/Elev= 30
       0 2530.95    12.1 2528.27    32.6 2521.63    39.4 2520.78    42.9 2519.76
    52.7 2515.83    72.6 2504.86    78.3 2503.15    95.4 2499.58   119.9  2497.6
   138.1 2497.38   146.6 2497.91   160.9 2500.29   197.8 2501.16   203.5 2500.88
   223.4 2498.38   285.3 2500.04   289.4 2499.48   300.82496.394   309.6 2495.57
   325.62497.354   341.9 2500.69   362.1  2506.4   379.8 2509.46   406.4 2505.85
   426.6 2504.93   454.8 2502.36   458.8 2502.14   469.3 2502.98   489.8 2502.66
#Mann= 5 ,-1,0
       0      .1       0   300.8    .045       0   325.6      .1       0
  377.09     .06       0  477.09      .1       0
Bank Sta=300.8,325.6
XS Rating Curve= 0 ,0
Exp/Cntr(USF)=0,0
Exp/Cntr=0.3,0.1

Type RM Length L Ch R = 1 ,68888   ,218.9,202.3,180.9
XS GIS Cut Line= 5
2215395.23599087648188.7913228722215528.32440056648367.999478503
2215507.24108814648446.403046591 2215510.5353557648523.488907653
2215531.61866813648601.233622228
#Sta/Elev= 30
       0 2533.27    10.4 2529.37    35.4 2524.47    55.3 2518.62    68.7 2516.12
    80.2 2511.16    89.6 2505.44    92.4 2504.26   100.1 2502.75   108.9  2500.2
     130 2498.07   163.9 2496.05   182.7  2498.2   201.1 2497.72   223.2 2499.07
   261.7 2498.04     270 2496.97     2942495.254   303.1 2494.53   311.2 2494.85
   323.1 2494.47   323.62494.514   327.2 2494.81   339.2 2497.47   348.2 2498.36
   363.2 2498.01   420.1 2498.24   441.3 2499.17   449.6 2499.07   462.1 2499.97
#Mann= 5 ,-1,0
       0      .1       0     294    .045       0   323.6      .1       0
  344.41     .06       0  451.57      .1       0
Bank Sta=294,323.6
XS Rating Curve= 0 ,0
Exp/Cntr(USF)=0,0
Exp/Cntr=0.3,0.1

Type RM Length L Ch R = 1 ,68686   ,138.7,144.1,147.1
XS GIS Cut Line= 3
2215217.26745104648486.2631194552215278.72429454  648507.9537701
2215646.65693355648660.906925572
#Sta/Elev= 30
       0 2535.24    23.4 2534.43      37 2531.25    48.5  2530.6    54.7 2528.82
    62.5 2528.04    75.4 2523.35    84.1 2521.28   100.9 2513.41   127.4 2494.45
   133.32493.219     149 2491.45     162 2492.12   166.4 2492.91     175 2494.34
   196.7 2493.04   209.7  2495.6   220.2 2495.42   231.4 2494.11   250.8 2493.61
     260 2494.45   274.7 2496.97     292  2496.2     357 2500.69   400.3  2501.7
   404.6 2503.25   413.3 2507.78     422 2510.69   443.5 2513.95   463.6 2518.22
#Mann= 4 ,-1,0
       0      .1       0   133.3    .045       0   166.4      .1       0
  405.17     .06       0
Bank Sta=133.3,166.4
XS Rating Curve= 0 ,0
Exp/Cntr(USF)=0,0
Exp/Cntr=0.3,0.1
